--- LtleHufCr.prj (project) ---

Proj Title=LtleHufCr
Current Plan=p01
Default Exp/Contr=0,0
English Units
Geom File=g01
Flow File=f01
Plan File=p01
BEGIN DESCRIPTION:
END DESCRIPTION:
DSS Export Rating Curves= 0
DSS Export Rating Curve Sorted= 0
DSS Export Volume Flow Curves= 0
DXF OffsetX= 0
DXF OffsetY= 0
DXF ScaleX= 0
DXF ScaleY= 0

--- LtleHufCr.p01 (plan) ---

Plan Title=Floodplain
Program Version=4.00
Geom File=g01
Flow File=f01
K Sum by GR=0
Std Step Tol=0.01
Critical Tol=0.01
Num of Std Step Trials=20
Max Error Tol=0.3
Flow Tol Ratio=0.001
Split Flow NTrial=30
Split Flow Tol=0.02
Split Flow Ratio=0.02
Log Output Level=0
Friction Slope Method=1
Unsteady Friction Slope Method=2
Unsteady Bridges Friction Slope Method=1
Global Log Level=0
CheckData=False
Run HTab=0
Run UNet=0
Run PostProcess=0
UNET Theta=0
UNET Theta Warmup=0
UNET ZTol=0
UNET ZSATol=0
UNET MxIter=0
UNET MaxInSteps=0
UNET DtIC=0
UNET DtMin=0
UNET MaxCRTS=0
UNET WFStab=0
UNET SFStab=0
UNET WFX=0
UNET SFX=0
UNET DSS MLevel=0
UNET DZMax Abort=0
UNET Convert EG Bridges=0
UNET Use Existing IB Tables=0
UNET Froude Limit=0
UNET Froude Power=0
Write IC File=0
Echo Input=False
Echo Output=False
Write Detailed=0

--- LtleHufCr.f01 (steady flow) ---

Flow Title=NFF Regression Equation
Program Version=4.00
Number of Profiles=1
Profile Names=P100yr
River Rch & RM=LtleHufCr,Main      ,10332.9
553.2813
River Rch & RM=LtleHufCr,Main      ,9872.9
571.1730
River Rch & RM=LtleHufCr,Main      ,9439.4
722.0478
River Rch & RM=LtleHufCr,Main      ,8244.6
755.4429
River Rch & RM=LtleHufCr,Main      ,7927.3
828.4366
River Rch & RM=LtleHufCr,Main      ,5817.5
864.7729
River Rch & RM=LtleHufCr,Main      ,5515.6
988.2262
River Rch & RM=LtleHufCr,Main      ,3365.9
1020.906
River Rch & RM=LtleHufCr,Main      ,2646.3
1141.506
River Rch & RM=LtleHufCr,Main      ,907.9
1214.717
River Rch & RM=LtleHufCr,Main      ,519.3
1220.268
Boundary for River Rch & Prof#=LtleHufCr,Main      ,1
Up Type=0
Dn Type=3
Dn Slope=0.021631

--- LtleHufCr.g01 (geometry) ---

Geom Title=USGS 10m DEM
Program Version=4.00

River Reach=LtleHufCr       ,Main
Reach XY= 30
     1769817.574      192435.934     1769528.691      192890.627
     1769442.041       192814.86     1769311.856      192837.046
     1769124.659      193002.031     1768689.398      193101.601
     1768619.073      193207.089     1768364.879      193229.828
     1768274.984      193324.715     1768192.938      193261.925
     1768048.417      193335.543      1767974.01      193266.111
     1767726.199      193391.691     1767180.194      193090.695
     1766009.832      193433.073     1765930.717      193682.696
     1765710.421      193838.199     1765519.453      194257.646
     1765299.158      194497.721     1765278.225      194654.608
     1765171.901      194663.398     1765218.678      194856.468
     1765138.199      195196.801     1764966.328      195238.404
     1764843.718      195675.992     1764369.639      196050.459
     1764008.077      196088.895     1763902.362      196327.605
     1763449.495      196509.025     1762873.792      196952.068

Type RM Length L Ch R = 1 ,10332.9 ,179.4,189.2,197.1
XS GIS Cut Line= 4
     1769422.612       192268.98      1769677.85      192426.474
     1769913.561       192482.33     1770194.219      192555.565
#Sta/Elev= 30
       0 1543.27      20  1542.6      40 1543.59      85 1542.11     125  1535.3
     140  1530.6     170 1516.42     195 1503.39   249.9 1469.48   269.9 1459.74
   289.9 1451.78   304.9 1448.48   364.2 1444.07   388.9 1438.65   428.2 1439.31
   438.3 1438.03   443.2 1438.41     468 1445.76   502.6 1464.52   522.4 1476.96
   537.2 1482.15   556.9 1496.56   655.2 1560.54   724.1 1601.25   753.6 1616.81
   792.9  1644.6   802.7 1649.12   817.5 1650.96   822.4 1652.83   832.2 1660.32
#Mann= 3 , 0 , 0
       0      .1       0   428.2    .045       0   443.2      .1       0
Bank Sta=428.2,443.2
XS Rating Curve= 0 ,0
Exp/Cntr=0.3,0.1

Type RM Length L Ch R = 1 ,10143.8 ,277.1,270.9,277.3
XS GIS Cut Line= 4
     1769391.469      192342.245     1769639.345      192539.583
     1769819.837      192655.098     1770091.778      192746.547
#Sta/Elev= 30
       0  1505.7    39.6 1496.05   108.9 1485.03   173.3 1476.89   193.1 1477.16
   237.6 1469.07     302 1461.33   321.8 1456.26   336.8 1446.72   346.7 1441.86
   366.7 1436.52   386.6 1435.16   388.9 1435.22   403.9 1435.77   446.4 1436.49
   456.4 1437.53   476.3 1443.16   496.2 1451.05   516.2 1463.98     541 1477.44
   550.9 1487.34   560.8 1495.58   630.1 1541.24   684.5 1579.41   773.5 1644.31
   778.5  1647.1   793.3 1648.17   808.1 1657.11   813.1 1662.59     818 1669.52
#Mann= 3 , 0 , 0
       0      .1       0   388.9    .045       0   403.9      .1       0
Bank Sta=388.9,403.9
XS Rating Curve= 0 ,0
Exp/Cntr=0.3,0.1

Type RM Length L Ch R = 1 ,9872.9  ,132.6,298.3,189.6
XS GIS Cut Line= 4
     1769295.388      192436.563     1769530.495      192736.706
     1769665.262      192909.979     1769908.325      193006.241
#Sta/Elev= 30
       0 1543.66    49.5 1530.22    79.2 1523.13      99 1516.74   113.9 1512.88
   153.5 1498.95   178.2 1487.34     208 1474.63   242.6  1463.3   341.6 1442.56
   386.2 1434.74   396.2  1432.3   411.2 1430.55   421.2 1430.35   446.1 1431.48
   480.6 1431.02   495.6 1430.97     511 1431.96   550.9 1431.83   605.7 1433.08
     655 1441.24   704.4 1444.39     734 1454.79   758.6 1466.04   768.5 1469.09
   783.3 1471.89   788.2 1473.53   827.7 1488.71   842.5 1495.12   862.2 1502.04
#Mann= 3 , 0 , 0
       0      .1       0   480.6    .045       0   495.6      .1       0
Bank Sta=480.6,495.6
XS Rating Curve= 0 ,0
Exp/Cntr=0.3,0.1

Type RM Length L Ch R = 1 ,9574.6  ,104.9,135.2,142.3
XS GIS Cut Line= 4
     1769356.795      192524.725     1769490.499      192747.123
     1769478.585      192992.027     1769568.189      193188.156
#Sta/Elev= 30
       0 1518.34    34.9 1508.62    59.9 1499.84    74.8 1491.92    99.8 1481.54
   109.8 1475.97   139.7 1466.17   184.6 1453.47   244.5 1438.08   269.3  1432.5
     284 1430.77     338 1427.87   372.3 1427.94   385.2 1429.57   400.2 1430.03
   426.2 1430.48   465.5 1433.74   480.2 1435.66   504.7 1441.28     539 1440.71
   573.3 1443.93   583.1 1447.51   602.7 1457.48   627.2 1463.65   646.8 1470.23
   656.6 1474.59   695.8 1495.36   705.6 1498.14   715.4 1497.64   720.3 1499.25
#Mann= 3 , 0 , 0
       0      .1       0   385.2    .045       0   400.2      .1       0
Bank Sta=385.2,400.2
XS Rating Curve= 0 ,0
Exp/Cntr=0.3,0.1

Type RM Length L Ch R = 1 ,9439.4  ,370.3,333.1,324.5
XS GIS Cut Line= 4
     1769292.765       192430.96      1769400.48      192710.057
     1769395.185      192984.084     1769431.192       193281.09
#Sta/Elev= 30
       0 1544.06    44.9 1541.72    89.8  1537.2   104.7 1534.88   119.7 1529.54
   144.6 1523.28   169.5 1513.98   229.4 1483.02   269.2  1465.8   324.1 1447.23
   363.9 1431.47   388.9 1425.68   402.1 1427.05   417.1 1428.32   563.3 1428.04
   598.2 1437.03   623.1 1442.06     648 1445.33     673 1451.76   692.9  1459.4
   702.9 1465.01   732.8 1491.25   737.8 1494.11   742.8  1495.4   752.8 1495.84
   757.7 1497.64   762.7  1500.8   787.6 1519.68   837.5    1551   872.4 1574.63
#Mann= 3 , 0 , 0
       0      .1       0   402.1    .045       0   417.1      .1       0
Bank Sta=402.1,417.1
XS Rating Curve= 0 ,0
Exp/Cntr=0.3,0.1

Type RM Length L Ch R = 1 ,9106.3  ,386.8,392.7,394.5
XS GIS Cut Line= 3
     1768897.443      192609.327     1769114.115      192954.035
     1769329.647      193317.309
#Sta/Elev= 30
       0 1668.75    14.9 1664.05    19.9 1661.56    54.6 1640.07    94.3 1607.24
   119.2 1588.73     149 1565.06   193.6 1532.39   243.3 1497.52     293 1467.02
   312.8 1457.98   342.6 1448.28   372.4 1436.99   412.1  1425.8   422.1 1423.98
   440.3 1424.77   455.3 1425.01   491.6 1426.05   516.5 1432.96   566.2 1439.74
     596 1446.07   620.8 1452.96   635.7  1461.8   650.6    1469   680.5  1488.1
   685.4 1490.46   695.4 1491.94   700.3  1493.8   720.2 1509.22   829.6 1574.16
#Mann= 3 , 0 , 0
       0      .1       0   440.3    .045       0   455.3      .1       0
Bank Sta=440.3,455.3
XS Rating Curve= 0 ,0
Exp/Cntr=0.3,0.1

Type RM Length L Ch R = 1 ,8713.6  ,469.4,469,470.2
XS GIS Cut Line= 3
     1768674.884      192684.042     1768783.914      193075.817
     1768932.027      193486.694
#Sta/Elev= 30
       0 1670.15     9.9 1667.42    24.8 1664.88    34.7 1659.85    89.3 1617.05
   158.7 1561.09   203.3 1527.77   233.1 1502.12   277.7 1471.57   307.5 1448.89
   317.4 1443.57   337.2 1436.14   357.1 1424.58     362 1422.87   381.9 1420.94
   399.2 1421.85   414.2 1422.78   456.3 1422.72   530.7 1424.74   555.6 1424.05
   590.3 1424.92   595.3 1426.07   605.2 1430.34   620.1 1438.41   654.8 1462.38
   679.6 1474.36   744.2 1514.68   754.1 1521.31   778.9 1540.15   843.4 1586.95
#Mann= 3 , 0 , 0
       0      .1       0   399.2    .045       0   414.2      .1       0
Bank Sta=399.2,414.2
XS Rating Curve= 0 ,0
Exp/Cntr=0.3,0.1

Type RM Length L Ch R = 1 ,8244.6  ,303.2,317.3,310.9
XS GIS Cut Line= 3
     1768269.991      192821.929     1768385.779      193226.744
     1768499.756      193624.412
#Sta/Elev= 30
       0 1561.55    34.7 1551.58    69.4 1539.73    89.2  1529.4   138.7 1506.35
   153.6 1500.33   168.4  1492.8   198.1 1481.53   257.6 1453.82   312.1 1435.16
   341.8  1422.5   376.5 1418.29   410.4 1417.07     421  1415.8   425.4 1416.05
   480.9 1424.32   500.8 1422.18   545.6 1423.42   565.6 1424.74   590.5 1429.06
   625.4  1429.3   630.4 1429.99   645.3 1434.82   665.3 1438.44   675.2 1439.07
   690.2 1437.84   705.1 1438.48   725.1 1437.72   794.8 1440.91   834.7 1444.18
#Mann= 3 , 0 , 0
       0      .1       0   410.4    .045       0   425.4      .1       0
Bank Sta=410.4,425.4
XS Rating Curve= 0 ,0
Exp/Cntr=0.3,0.1

Type RM Length L Ch R = 1 ,7927.3  ,420.1,415.8,412.2
XS GIS Cut Line= 3
     1768124.351      192847.202     1768184.029      193257.467
     1768256.591      193688.719
#Sta/Elev= 30
       0 1617.42      25 1596.72      40 1585.44    79.9 1556.68    94.9 1547.21
   124.9 1526.34   144.8 1509.53   164.8 1494.58   239.8 1449.73   264.7 1439.49
   289.7  1432.5   314.7 1429.48   344.6 1416.28   364.6 1415.25   374.6 1412.56
   415.9 1413.99   430.9 1414.41   454.3 1414.14   494.1 1411.68   533.8 1412.44
   578.6 1416.47   608.4 1425.47   618.3 1427.26   653.1 1430.11     678 1434.42
   707.8 1435.32   737.6 1441.95   757.5 1448.02   807.2 1465.18   851.9 1483.95
#Mann= 3 , 0 , 0
       0      .1       0   415.9    .045       0   430.9      .1       0
Bank Sta=415.9,430.9
XS Rating Curve= 0 ,0
Exp/Cntr=0.3,0.1

Type RM Length L Ch R = 1 ,7511.5  ,373.9,391.5,405.8
XS GIS Cut Line= 3
     1767756.751      192912.987     1767854.457      193347.321
     1767941.437      193747.448
#Sta/Elev= 30
       0 1589.54    34.6  1572.5    69.2 1552.08   108.8 1524.01   143.4 1500.87
   202.8 1467.96   222.6 1457.92     277 1440.82   296.8 1438.44   321.5 1432.61
   326.5 1430.03   346.3 1415.11   356.2 1410.53     366 1408.82   405.6 1408.04
   420.5 1406.37   437.7 1408.05   452.7    1409   510.1 1408.94   525.1 1412.09
     560 1423.92     575 1426.67     595 1433.44     630 1435.94   644.9 1443.02
   694.9 1462.91   734.8 1480.81   774.8 1501.26   829.7  1534.1   854.7 1547.74
#Mann= 3 , 0 , 0
       0      .1       0   437.7    .045       0   452.7      .1       0
Bank Sta=437.7,452.7
XS Rating Curve= 0 ,0
Exp/Cntr=0.3,0.1

Type RM Length L Ch R = 1 ,7120    ,163.9,169.1,174.5
XS GIS Cut Line= 4
     1767656.339      192906.115     1767555.665       193257.38
     1767499.403      193386.313     1767295.459      193669.558
#Sta/Elev= 30
       0 1588.34    14.8 1580.75    39.5 1564.74    74.1 1549.31   153.1  1503.9
   192.6 1482.49   212.3 1473.88   246.9 1456.14   281.5 1441.16     316 1424.36
   345.7 1418.23   360.5 1413.38   375.1 1407.01   394.5 1402.45   408.2  1403.6
   423.2 1404.85   467.3 1408.78   486.7 1415.27   506.1 1423.68     516  1426.2
     546 1429.95   590.8 1431.94   620.8 1436.22   635.7 1439.45   665.6 1442.05
   690.6  1445.3   750.4 1455.06   815.2 1468.07   835.2 1470.56   855.1 1474.32
#Mann= 3 , 0 , 0
       0      .1       0   408.2    .045       0   423.2      .1       0
Bank Sta=408.2,423.2
XS Rating Curve= 0 ,0
Exp/Cntr=0.3,0.1

Type RM Length L Ch R = 1 ,6950.9  ,76.4,73.4,70.4
XS GIS Cut Line= 4
     1767551.213      192924.757     1767422.411       193180.73
     1767350.673      193280.185     1767268.083      193564.844
#Sta/Elev= 30
       0 1567.64    19.8    1554    39.5 1538.68    74.1 1513.14   108.7 1489.12
   133.4 1474.15   158.1 1457.59   172.9 1449.67   237.2 1437.96   276.7 1428.64
   291.5 1422.86   325.8 1406.15   343.1 1404.11   358.1 1401.81     365 1401.19
   369.9 1401.98   374.8 1403.82   399.4 1414.79   404.3 1416.42   428.9 1422.18
   443.8 1423.73   473.4  1424.1   488.2 1424.98   537.6 1428.82   547.5 1430.43
   577.1 1437.08   631.5  1445.1   666.1  1451.6   680.9 1455.02   705.6 1468.26
#Mann= 3 , 0 , 0
       0      .1       0   343.1    .045       0   358.1      .1       0
Bank Sta=343.1,358.1
XS Rating Curve= 0 ,0
Exp/Cntr=0.3,0.1

Type RM Length L Ch R = 1 ,6877.5  ,78.6,72.7,66.9
XS GIS Cut Line= 4
     1767525.381      192887.206     1767380.173      193101.197
     1767303.748      193236.215     1767268.083      193496.061
#Sta/Elev= 30
       0 1574.17    14.9 1567.87    44.8 1549.85    89.5 1519.37   104.4 1507.19
   124.3 1492.58   134.3 1486.05   139.2 1483.52   149.2 1478.65   159.1 1474.67
   198.9 1462.53   292.6 1424.98   302.2  1419.6   316.8 1409.88   321.6 1407.38
   339.8 1403.94   354.8 1401.36   355.6 1401.24   365.3 1402.08     375 1405.53
   389.5 1412.19   394.4 1413.08   408.9 1412.89   443.4  1415.2   478.1 1418.61
   527.6  1425.1   557.3 1426.68     587 1431.08   601.8 1435.28     676 1446.83
#Mann= 3 , 0 , 0
       0      .1       0   339.8    .045       0   354.8      .1       0
Bank Sta=339.8,354.8
XS Rating Curve= 0 ,0
Exp/Cntr=0.3,0.1

Type RM Length L Ch R = 1 ,6804.8  ,71,69.8,68.6
XS GIS Cut Line= 4
     1767466.789      192854.089     1767319.033      193045.152
     1767252.798      193238.762     1767212.038      193536.821
#Sta/Elev= 30
       0 1573.13     9.9 1568.17    39.4 1550.39    64.1 1539.85    98.6 1523.68
   123.2 1509.63     143 1496.89   162.7  1485.9     212  1461.5   256.5 1436.25
   281.5 1416.01   291.4 1409.23   301.4 1405.52   312.9 1403.87   316.4 1403.51
   327.9 1404.26   336.4 1405.42   346.3 1405.53   371.3 1410.34   391.3  1410.3
   431.2 1411.99   515.2  1419.2   544.8  1423.5   564.5 1423.91   584.2 1426.95
   608.9 1428.35   648.4 1437.58     673 1445.57   697.7 1457.12     747 1482.29
#Mann= 3 , 0 , 0
       0      .1       0   312.9    .045       0   327.9      .1       0
Bank Sta=312.9,327.9
XS Rating Curve= 0 ,0
Exp/Cntr=0.3,0.1

Type RM Length L Ch R = 1 ,6735    ,83.2,75.5,67.8
XS GIS Cut Line= 4
     1767415.838      192818.424      1767250.25      193009.487
     1767201.848      193243.858     1767176.372      193508.798
#Sta/Elev= 30
       0 1593.68    19.8 1580.47    34.7 1572.03    64.4 1559.57   104.1 1544.41
   183.4 1504.44   203.3    1491   213.2 1482.52     233 1463.09   262.8 1436.35
   277.8 1425.07   287.7 1419.49   302.7 1414.19   322.6  1403.4   330.6  1401.4
   342.6 1399.72   345.6 1400.01   362.5 1403.64   382.5 1404.98   407.4 1409.01
   432.3 1409.22   477.2 1412.18   566.1 1420.59   600.6 1422.46   615.4 1426.09
     645 1428.74   654.8 1431.56   679.4 1441.04   718.9 1458.62   758.3  1481.1
#Mann= 3 , 0 , 0
       0      .1       0   330.6    .045       0   345.6      .1       0
Bank Sta=330.6,345.6
XS Rating Curve= 0 ,0
Exp/Cntr=0.3,0.1

Type RM Length L Ch R = 1 ,6659.5  ,69.2,66.7,64.3
XS GIS Cut Line= 4
     1767357.013      192757.438     1767151.763      193050.298
     1767169.698       193180.73     1767113.853      193558.016
#Sta/Elev= 30
       0 1636.97    49.7 1608.92    94.4 1579.96   134.1 1560.84   163.9 1544.73
   193.7 1524.53   218.6 1509.68   278.2 1481.28     303 1467.79   312.9 1461.41
   332.8 1446.15   386.9 1402.55   391.8 1400.55   394.1 1400.53   396.6 1400.52
   409.1 1401.22   425.9 1403.05   450.3 1403.53   479.5 1408.48   528.9 1410.99
   603.2 1416.64   642.8  1421.9   667.6 1426.29   692.4 1427.54   707.2 1434.62
   722.1 1439.88   741.9 1448.35   766.7 1459.93   806.3 1481.22   870.7 1518.27
#Mann= 3 , 0 , 0
       0      .1       0   394.1    .045       0   409.1      .1       0
Bank Sta=394.1,409.1
XS Rating Curve= 0 ,0
Exp/Cntr=0.3,0.1

Type RM Length L Ch R = 1 ,6592.7  ,56.6,58.3,61.5
XS GIS Cut Line= 4
     1767054.092      192747.093     1767071.925      193022.224
     1767125.422      193236.215     1767094.852      193552.106
#Sta/Elev= 30
       0 1615.94    29.5 1594.81    59.1 1575.01    98.5 1550.35   177.2 1498.51
   196.9 1487.79   236.3 1469.42   260.9 1455.81   270.8 1449.68     310 1419.94
   324.7 1409.92   329.6 1407.44     348 1401.19   354.1 1399.49     363 1398.69
   363.9 1398.67   383.6 1401.79   417.9 1401.17   437.5 1402.36   506.2 1411.24
   550.8 1414.44   595.5  1421.9   615.3 1425.98   630.2 1426.75   640.1 1428.67
   659.9 1437.61   689.7 1450.01   709.5 1459.44   764.1 1490.18   813.6 1519.85
#Mann= 3 , 0 , 0
       0      .1       0     348    .045       0     363      .1       0
Bank Sta=348,363
XS Rating Curve= 0 ,0
Exp/Cntr=0.3,0.1

Type RM Length L Ch R = 1 ,6534.4  ,243.5,241.8,238.8
XS GIS Cut Line= 4
     1766967.477      192759.831      1767026.07      193060.437
     1767079.567      193315.188     1767059.187      193567.391
#Sta/Elev= 30
       0 1599.71     9.9 1591.22    34.6 1574.64      79 1546.44   133.4 1514.42
     163 1489.07   197.6 1468.03   212.4 1457.23   217.4 1454.52     242 1445.94
   266.8 1432.06   291.4    1425     321 1406.77   335.7 1402.38     361 1399.31
     375 1397.77     376 1397.96   389.8 1401.08   414.3 1400.51   463.4  1402.1
   522.4 1408.93   546.9 1414.42   581.4 1418.82   621.1 1427.87     641 1437.92
   675.7 1451.34   705.5 1467.19   735.2 1485.14   750.1 1492.77   819.6  1535.2
#Mann= 3 , 0 , 0
       0      .1       0     361    .045       0     376      .1       0
Bank Sta=361,376
XS Rating Curve= 0 ,0
Exp/Cntr=0.3,0.1

Type RM Length L Ch R = 1 ,6292.7  ,164.8,164.1,163.1
XS GIS Cut Line= 3
     1766739.938      192753.961     1766822.549      193158.006
      1766901.45       193567.33
#Sta/Elev= 30
       0 1502.52    29.8  1498.8    59.6 1493.38    99.4 1483.76   114.3 1479.39
   129.2 1472.94   173.9 1446.78   188.8 1438.98   198.8 1432.95   243.5  1413.4
   248.4 1412.21   303.1 1405.21     323 1404.07   362.7 1400.24   402.5 1398.19
   404.9 1398.28   419.9 1398.77   447.1 1399.16   457.1 1400.83     472 1404.59
   511.7 1409.68   571.2 1425.17   586.1 1431.83     601 1440.25   630.8 1454.01
   680.4 1480.43   744.9 1511.53   759.8 1520.38   799.5 1546.42   829.3 1564.57
#Mann= 3 , 0 , 0
       0      .1       0   404.9    .045       0   419.9      .1       0
Bank Sta=404.9,419.9
XS Rating Curve= 0 ,0
Exp/Cntr=0.3,0.1

Type RM Length L Ch R = 1 ,6128.6  ,312.6,311,309.7
XS GIS Cut Line= 4
     1766467.665      192868.055     1766645.757      193095.465
     1766697.814      193314.654     1766730.693      193580.422
#Sta/Elev= 30
       0 1423.11    94.6 1421.65   149.4 1417.04   189.2 1414.86   204.2 1412.66
   219.1 1411.65     244  1408.7   313.3  1403.3   352.5 1396.71   388.2 1395.91
   391.7 1395.86   403.2 1396.19   411.3 1397.49     426 1404.12   435.8 1407.47
   450.5 1409.83     470 1417.67   479.8 1420.32   489.6 1421.74   519.1 1422.88
     524 1424.55   543.9 1436.31   568.7 1446.24   593.5 1457.43   608.4 1465.31
     658 1496.03   667.9 1502.82   707.5 1532.17   732.3 1549.02   781.9 1584.29
#Mann= 3 , 0 , 0
       0      .1       0   388.2    .045       0   403.2      .1       0
Bank Sta=388.2,403.2
XS Rating Curve= 0 ,0
Exp/Cntr=0.3,0.1

Type RM Length L Ch R = 1 ,5817.5  ,328.1,301.9,289.6
XS GIS Cut Line= 3
     1766248.476      192884.495     1766375.495       193285.94
     1766492.836      193677.646
#Sta/Elev= 30
       0 1476.31    24.8 1457.43    34.7 1452.95    44.6 1450.98    69.4 1450.57
    79.3 1447.97   118.9 1421.17   133.8 1414.15   148.6 1412.44   168.4 1407.73
   307.1 1400.95   336.8 1393.34   371.5 1390.09   401.2  1391.4   408.8 1390.81
   416.1 1390.11   423.8 1392.71     446 1402.93   470.9 1415.88   485.9 1420.85
   535.8 1421.82   540.7    1423   560.7 1436.18   585.6 1447.43   605.6 1458.25
   650.4 1490.67   665.4 1499.73   735.2 1546.13   760.2 1561.05     830 1605.22
#Mann= 3 , 0 , 0
       0      .1       0   408.8    .045       0   423.8      .1       0
Bank Sta=408.8,423.8
XS Rating Curve= 0 ,0
Exp/Cntr=0.3,0.1

Type RM Length L Ch R = 1 ,5515.6  ,459.8,459.6,460.4
XS GIS Cut Line= 4
     1765771.412      193152.396     1766034.766      193328.354
     1766179.979      193465.347     1766351.517      193748.446
#Sta/Elev= 30
       0  1581.6     9.9 1575.39    14.8 1571.38    44.5 1553.67   103.9 1510.99
   153.4 1479.62   183.1 1459.41     193 1453.22   212.8 1443.13   232.6 1429.31
   267.2 1408.52   282.1 1402.56   301.9  1396.9   336.7 1394.64   361.6 1389.71
   391.6 1389.17   397.7 1389.23   412.7 1389.57   426.5  1389.2   456.5 1392.43
   516.4 1423.36   536.1 1426.03   541.1 1427.93   565.8 1440.61   620.1 1456.79
   659.6 1471.51   694.2 1487.71   723.9 1503.46     793 1543.38   847.4 1575.84
#Mann= 3 , 0 , 0
       0      .1       0   397.7    .045       0   412.7      .1       0
Bank Sta=397.7,412.7
XS Rating Curve= 0 ,0
Exp/Cntr=0.3,0.1

Type RM Length L Ch R = 1 ,5056    ,410,405.4,400.9
XS GIS Cut Line= 3
     1765554.523      193471.867     1765882.801      193751.592
     1766198.093       194006.83
#Sta/Elev= 30
       0 1510.21    19.8 1500.16    34.7 1490.72    94.2 1465.51     119  1452.1
   143.8 1442.57   178.5 1436.87   218.1  1426.1     233 1424.05   257.8 1422.47
   292.5 1422.92   337.1 1416.05     347 1413.15   371.8 1391.12   381.7 1385.27
   387.5  1383.5   402.5  1383.2   406.5 1383.16   431.3 1388.15     461 1390.88
   500.6 1407.96   525.3 1409.46   535.2 1412.24   559.9 1426.98   574.8 1432.66
   624.2 1461.84   673.7  1488.4   728.1 1522.18   802.3 1565.85     837 1589.12
#Mann= 3 , 0 , 0
       0      .1       0   387.5    .045       0   402.5      .1       0
Bank Sta=387.5,402.5
XS Rating Curve= 0 ,0
Exp/Cntr=0.3,0.1

Type RM Length L Ch R = 1 ,4650.6  ,405.4,407.3,410.1
XS GIS Cut Line= 3
     1765265.087      193823.243     1765617.205      194033.244
     1765959.274      194258.209
#Sta/Elev= 30
       0  1565.2      10  1557.4      30 1544.35      65 1519.51     125 1475.66
     170  1448.4     180 1444.13     240  1425.3     250 1423.66     270 1422.66
     285 1418.77     330 1403.38     335 1400.88     355    1387     360 1384.93
     383  1382.4     398 1381.39     405 1381.27     415 1382.58     435 1388.97
   489.9  1392.2   514.8  1395.1   544.8 1401.82   574.8 1412.91   589.7 1414.62
   649.6 1448.38   699.6 1480.53   719.5 1490.27   754.5 1511.37   819.4 1545.94
#Mann= 3 , 0 , 0
       0      .1       0     383    .045       0     398      .1       0
Bank Sta=383,398
XS Rating Curve= 0 ,0
Exp/Cntr=0.3,0.1

Type RM Length L Ch R = 1 ,4243.3  ,536.4,529.9,522.6
XS GIS Cut Line= 3
      1765090.98      194146.636     1765426.905      194383.146
     1765743.448      194642.566
#Sta/Elev= 30
       0 1576.46    64.4 1528.22    89.1 1513.34   128.7 1486.03   153.4 1470.68
   163.3 1463.06   217.8 1431.08   237.6 1416.05   257.4 1409.46   287.1 1393.81
   316.8 1382.47   386.1 1378.36   394.2  1376.9   405.9 1375.09   409.2 1375.41
   425.8 1379.92   450.8 1388.79   465.7 1389.99   480.7 1393.88   495.7 1400.56
   525.6 1410.22   545.6 1418.69   560.6 1425.72   585.5 1440.91   605.5  1451.1
   640.4 1471.44   670.4 1486.52   730.3 1519.21   765.2 1537.16   820.1 1562.75
#Mann= 3 , 0 , 0
       0      .1       0   394.2    .045       0   409.2      .1       0
Bank Sta=394.2,409.2
XS Rating Curve= 0 ,0
Exp/Cntr=0.3,0.1

Type RM Length L Ch R = 1 ,3713.4  ,346.5,347.5,347.7
XS GIS Cut Line= 4
     1764782.303      194578.746     1765033.261      194685.403
     1765312.451      194766.965     1765670.066      194835.978
#Sta/Elev= 30
       0 1485.12    19.8 1479.36    64.4 1462.98   148.7 1427.37   173.5 1420.67
   203.3 1410.32   218.2    1407     238 1404.95   267.7 1397.64   282.5 1395.32
   326.9 1390.68   341.7 1390.74   351.6 1389.42   381.1  1382.4   405.5 1375.16
   415.6 1372.18   420.5 1372.15   435.4 1373.52   494.5 1372.38   504.4 1373.04
   509.3 1374.99     534 1391.25   553.7 1397.69   578.5 1403.29   603.5 1411.82
   628.4 1425.26   743.2  1491.6     838 1551.72   912.8 1602.26   927.8 1613.56
#Mann= 3 , 0 , 0
       0      .1       0   405.5    .045       0   420.5      .1       0
Bank Sta=405.5,420.5
XS Rating Curve= 0 ,0
Exp/Cntr=0.3,0.1

Type RM Length L Ch R = 1 ,3365.9  ,732.5,719.6,727.9
XS GIS Cut Line= 3
     1764759.403      194904.678     1765212.463      195063.896
     1765582.545      195183.241
#Sta/Elev= 30
       0 1473.25    14.8 1470.55    44.6 1461.03    74.3  1449.9   108.9  1436.4
   133.7 1423.31   183.2 1402.07   207.9 1392.58   222.8 1388.38   252.5 1384.29
   292.1 1381.44   321.8 1377.73   361.4 1369.11   391.1 1369.18   427.4 1365.68
   430.7 1365.62   442.4 1367.04   455.5 1369.69   495.2 1390.66   525.1 1400.74
     560 1414.21   619.8 1441.59   644.7 1454.02   669.7  1462.4   684.6 1470.26
   704.6 1477.16   724.5 1485.35   779.3 1512.24   849.1 1543.66   869.1 1550.93
#Mann= 3 , 0 , 0
       0      .1       0   427.4    .045       0   442.4      .1       0
Bank Sta=427.4,442.4
XS Rating Curve= 0 ,0
Exp/Cntr=0.3,0.1

Type RM Length L Ch R = 1 ,2646.3  ,244.4,249.7,254.9
XS GIS Cut Line= 4
     1764506.385      195390.593      1764829.42      195550.392
     1764975.299       195648.92       1765262.4       195739.42
#Sta/Elev= 30
       0 1559.84    19.8    1544    59.2 1518.79    88.9 1504.28   148.1 1479.64
   177.7 1461.87   187.6 1457.02   217.2 1437.13   241.9 1418.81   271.5 1401.25
   286.3 1394.44   325.8 1380.74   365.3 1360.43     380 1358.25   397.8 1358.17
   412.8 1356.15   414.2 1355.99   438.6 1360.64   458.2 1360.29     468    1361
   507.1 1367.35   526.6 1371.72   551.2 1374.43   595.6 1388.83   659.8 1407.26
   679.5 1413.83   753.6 1442.05   788.1 1457.26   807.8  1465.1   837.5 1475.31
#Mann= 3 , 0 , 0
       0      .1       0   397.8    .045       0   412.8      .1       0
Bank Sta=397.8,412.8
XS Rating Curve= 0 ,0
Exp/Cntr=0.3,0.1

Type RM Length L Ch R = 1 ,2396.7  ,72.2,73.1,72.4
XS GIS Cut Line= 4
      1764532.18      195478.426     1764697.331      195725.264
     1764800.328      195838.916     1764995.668      196044.911
#Sta/Elev= 30
       0 1505.54     9.9 1502.12    39.6 1494.89    59.4 1485.15   108.9 1455.23
   173.2 1409.87     193 1398.02   202.9 1393.53   212.8 1390.99   247.5 1386.07
   277.2 1365.86   287.1 1360.19     297  1356.8   306.9 1356.26     357 1357.86
     372 1357.59     396  1357.6   410.8 1359.38   430.6 1366.57   450.4 1376.68
   460.3 1380.11   475.3 1381.98   520.1 1391.92   559.9 1397.91   579.9 1404.07
   619.7 1420.02   659.6 1431.65   694.4 1439.68   724.3 1448.68   734.3 1452.88
#Mann= 3 , 0 , 0
       0      .1       0     357    .045       0     372      .1       0
Bank Sta=357,372
XS Rating Curve= 0 ,0
Exp/Cntr=0.3,0.1

Type RM Length L Ch R = 1 ,2323.6  ,28.8,29.5,31.8
XS GIS Cut Line= 4
     1764478.906       195510.39     1764652.936      195767.883
     1764768.364      195902.846     1764921.084        196075.1
#Sta/Elev= 30
       0 1511.83    14.8 1503.64    34.5 1494.29    44.4 1491.09    59.2 1484.96
    88.8 1470.47   118.4 1452.95   143.1 1436.78   172.7 1414.23   197.3 1398.01
   212.1 1392.38   251.6  1381.7   276.3 1369.22     296 1356.78   300.9 1355.62
   320.6 1355.62   337.4 1354.32   345.3 1352.42   350.2  1352.4   352.4 1352.65
   384.8 1358.56   414.4 1359.87     439 1366.27   458.8 1368.03   498.2 1374.21
   503.1 1375.65   586.3 1403.41   694.1 1453.26   708.8 1459.59   718.6 1462.64
#Mann= 3 , 0 , 0
       0      .1       0   337.4    .045       0   352.4      .1       0
Bank Sta=337.4,352.4
XS Rating Curve= 0 ,0
Exp/Cntr=0.3,0.1

Type RM Length L Ch R = 1 ,2294.1  ,45.4,44.4,43.5
XS GIS Cut Line= 4
       1764413.2      195540.579      1764596.11      195741.246
     1764738.175      195917.052     1764887.343      196096.409
#Sta/Elev= 30
       0 1522.86    44.4 1495.12      74 1481.65   103.7 1464.04   133.3  1445.4
   167.8 1419.38   177.7 1412.57   192.5 1403.85   217.2 1392.77   241.9 1384.54
   266.6 1380.44   276.4  1377.5   296.1 1365.17   310.8 1358.71   325.6 1355.41
   346.6 1354.18     355 1353.87   361.6 1354.02   384.5 1355.74   409.1 1360.55
   443.5 1363.33   507.5 1375.34   522.4 1375.56   527.3 1376.32   562.1 1385.06
   596.8 1395.14   651.4 1418.79   681.2 1435.47     706 1451.51   730.8 1462.48
#Mann= 3 , 0 , 0
       0      .1       0   346.6    .045       0   361.6      .1       0
Bank Sta=346.6,361.6
XS Rating Curve= 0 ,0
Exp/Cntr=0.3,0.1

Type RM Length L Ch R = 1 ,2249.6  ,47.5,43.4,43
XS GIS Cut Line= 4
     1764361.702      195593.854     1764581.903      195794.521
     1764697.331      195925.931     1764869.585      196123.047
#Sta/Elev= 30
       0 1512.77    14.9 1502.78    49.6 1482.49    74.5 1466.05    94.3 1455.83
   119.2 1440.28   158.9 1409.98   168.8 1404.46   188.7 1396.06   208.5 1389.16
   233.4 1384.98   268.1 1377.03   312.9 1357.74   317.9 1356.29   333.2 1355.03
   348.2 1354.28   352.9 1354.15   367.9 1355.21   397.9 1362.88   422.8 1365.14
   452.8 1371.75   507.4 1380.67   522.2 1381.98   556.8 1382.64   571.6 1386.46
   655.6 1416.18   680.3 1428.65   690.2 1435.13   709.9 1450.29   734.6 1462.94
#Mann= 3 , 0 , 0
       0      .1       0   333.2    .045       0   348.2      .1       0
Bank Sta=333.2,348.2
XS Rating Curve= 0 ,0
Exp/Cntr=0.3,0.1

Type RM Length L Ch R = 1 ,2206.2  ,54.1,60.3,62.5
XS GIS Cut Line= 3
     1764266.835      195608.553     1764585.121      195862.098
     1764876.786      196176.168
#Sta/Elev= 30
       0 1531.54   104.2 1468.95   148.9 1444.66   168.7 1432.06   223.3 1399.58
   238.2 1393.62     268 1387.49   287.8 1380.51   322.6  1370.3   332.5  1368.3
   362.3 1357.53   399.4 1352.54     402  1352.3   414.4 1353.08   436.8  1355.1
   461.8 1363.62   476.7 1365.81   506.6 1375.75   536.5 1382.88   586.4 1388.35
   626.2 1389.05   646.2 1390.98     681  1396.1   710.9 1403.82   735.9 1415.19
   770.8 1434.83   790.7 1451.18   795.7 1454.33   815.6 1465.63   835.5 1475.32
#Mann= 3 , 0 , 0
       0      .1       0   399.4    .045       0   414.4      .1       0
Bank Sta=399.4,414.4
XS Rating Curve= 0 ,0
Exp/Cntr=0.3,0.1

Type RM Length L Ch R = 1 ,2146    ,330.9,339.7,349.2
XS GIS Cut Line= 4
     1764287.118      195675.541     1764514.422      195856.674
     1764603.213      195973.878     1764750.605       196151.46
#Sta/Elev= 30
       0 1485.64    44.3 1459.25    73.9 1443.26   103.4  1426.1   152.7 1399.24
   162.6 1394.57   182.3 1387.96   187.2 1387.27     202 1387.48   211.8 1386.11
   231.5 1378.38   261.1  1371.6   285.7  1359.6   295.6 1356.72   320.1 1354.25
   344.6 1353.55   358.3 1351.82   364.2 1351.66   373.3 1353.69   398.5 1361.32
   403.4 1363.81   413.2  1370.5   432.8 1377.59   442.6 1379.95   506.4 1387.61
     531 1389.83   570.3 1395.04   594.8 1399.79   624.3 1403.02   668.5 1409.69
#Mann= 3 , 0 , 0
       0      .1       0   358.3    .045       0   373.3      .1       0
Bank Sta=358.3,373.3
XS Rating Curve= 0 ,0
Exp/Cntr=0.3,0.1

Type RM Length L Ch R = 1 ,1806.2  ,124,132.1,139.7
XS GIS Cut Line= 3
     1764170.141      195671.143     1764274.476      196090.295
     1764365.351      196485.522
#Sta/Elev= 30
       0 1514.34    54.6 1478.65    59.6  1475.1    79.4 1456.89    94.3  1447.7
   104.3 1442.32   129.1 1432.84   158.9 1418.76   208.5 1401.51   238.3 1393.86
   297.9 1380.85   312.8 1374.71   337.6 1361.14   357.5 1353.93   382.3 1350.86
   412.1 1350.56   424.4 1348.22   436.9 1346.76   439.4 1347.02   461.6 1349.46
   466.6 1351.04   496.2  1371.9     521 1386.76   575.4 1397.78   639.7 1408.37
   664.4 1415.99   679.2 1422.91   708.9 1439.75   748.5 1459.18   837.5 1509.12
#Mann= 3 , 0 , 0
       0      .1       0   424.4    .045       0   439.4      .1       0
Bank Sta=424.4,439.4
XS Rating Curve= 0 ,0
Exp/Cntr=0.3,0.1

Type RM Length L Ch R = 1 ,1674.2  ,306.2,271.2,244.6
XS GIS Cut Line= 4
     1763975.739      195694.354     1764156.096      195988.473
     1764133.898      196182.703     1764269.859      196501.795
#Sta/Elev= 30
       0 1542.45    78.9 1490.69   118.3 1463.15   147.9 1444.87   187.3 1418.36
   211.9 1404.45   226.7 1399.05   256.3 1393.98   290.8  1384.9   335.2 1378.92
     345 1375.42   384.1 1356.49   393.9 1352.84   413.4 1349.16   428.1 1348.43
   444.3 1348.96   459.3 1349.21   472.1 1348.85   481.9 1349.88   491.6 1353.28
   506.3 1361.01   545.5 1365.02   634.6 1378.01   659.4 1382.19   684.2 1389.18
     704 1396.52   728.8 1408.03   773.4 1432.43   862.6 1477.19   887.4 1491.33
#Mann= 3 , 0 , 0
       0      .1       0   444.3    .045       0   459.3      .1       0
Bank Sta=444.3,459.3
XS Rating Curve= 0 ,0
Exp/Cntr=0.3,0.1

Type RM Length L Ch R = 1 ,1403    ,92.3,94.3,92.8
XS GIS Cut Line= 4
     1763595.426      195980.533     1763856.427      196152.181
     1764075.629      196271.494     1764211.612      196537.798
#Sta/Elev= 30
       0 1521.72    49.6 1493.21     124 1447.86   173.6 1420.72   193.4 1408.54
   228.1 1390.65   257.8 1379.81   272.7 1376.31   332.4 1371.89   352.3 1368.66
   362.3    1364   382.3 1349.53   397.2 1344.76   397.2 1344.75   412.2 1343.56
   447.2 1343.07   457.1 1343.51     507 1354.95     537 1358.02     562 1363.01
   581.9 1369.03   621.8 1374.61   631.7 1377.55   646.7 1383.67   671.6 1391.75
   696.5 1403.38   751.3 1433.55   821.1 1468.19     846 1478.73     861 1488.06
#Mann= 3 , 0 , 0
       0      .1       0   397.2    .045       0   412.2      .1       0
Bank Sta=397.2,412.2
XS Rating Curve= 0 ,0
Exp/Cntr=0.3,0.1

Type RM Length L Ch R = 1 ,1308.7  ,48.1,49.2,54.3
XS GIS Cut Line= 4
     1763636.866      196039.112     1763869.102       196254.52
     1764010.463      196326.883     1764118.167      196486.756
#Sta/Elev= 30
       0 1473.89    14.8  1463.9    89.1 1419.23   153.4 1377.96   158.4 1377.16
   168.3 1373.86   202.9 1366.57   227.7 1363.62   262.3 1361.47   287.1 1357.93
   341.6 1344.56   371.6 1339.82   376.3 1338.69   381.3 1338.63   386.6 1339.43
   401.1 1341.69     421 1342.02   425.9 1343.37   445.8    1352   495.3 1368.81
     520 1372.36   529.9 1376.08   549.7 1381.88   579.4 1394.06   594.2 1398.44
   599.1  1400.5   618.9 1412.63   628.8 1420.49   633.7  1423.6   668.3 1442.97
#Mann= 3 , 0 , 0
       0      .1       0   371.6    .045       0   386.6      .1       0
Bank Sta=371.6,386.6
XS Rating Curve= 0 ,0
Exp/Cntr=0.3,0.1

Type RM Length L Ch R = 1 ,1259.5  ,40.9,48.5,55.7
XS GIS Cut Line= 4
     1763635.183      196060.989     1763845.542      196273.031
     1763986.903      196397.564     1764089.558      196515.365
#Sta/Elev= 30
       0 1461.02    34.8 1438.88   109.5 1396.06   139.4 1380.75   154.3 1374.52
   169.2 1369.38   184.2 1365.44   209.1 1361.55   253.9 1357.64   273.8 1356.74
   288.7 1354.97   298.7 1352.91   323.5 1344.03   363.1 1341.75   370.3 1340.09
     383  1337.6   385.3 1338.03   412.7 1345.27   417.7 1347.17   427.6  1353.4
   437.5 1357.84   462.3  1364.5   477.2 1366.92   482.1 1368.42   487.1 1370.44
   501.7 1378.71   545.7 1396.36     575 1411.08   618.9  1439.5   643.3 1452.89
#Mann= 3 , 0 , 0
       0      .1       0   370.3    .045       0   385.3      .1       0
Bank Sta=370.3,385.3
XS Rating Curve= 0 ,0
Exp/Cntr=0.3,0.1

Type RM Length L Ch R = 1 ,1211.1  ,136.4,136.9,137.3
XS GIS Cut Line= 4
     1763599.842      196074.452     1763818.616      196267.982
     1763919.588      196449.733     1764054.218      196555.754
#Sta/Elev= 30
       0 1464.34    34.6  1443.4    94.1 1410.05   148.5 1382.77   188.1  1367.8
     198  1365.7   207.9  1365.7   247.5  1358.3   306.9 1353.22   311.9 1352.05
   331.7 1343.16   361.4 1341.99   370.7 1340.22   381.2 1337.74   385.7 1338.36
     401  1342.3   415.8 1344.48   435.6  1359.1   450.5 1365.91   475.2 1369.15
   485.2 1371.46   504.9 1380.79   514.7 1382.68   539.2  1390.9   553.9 1393.81
   563.6 1397.44   573.4 1402.88   617.5 1433.88   666.5 1460.28   671.4 1462.02
#Mann= 3 , 0 , 0
       0      .1       0   370.7    .045       0   385.7      .1       0
Bank Sta=370.7,385.7
XS Rating Curve= 0 ,0
Exp/Cntr=0.3,0.1

Type RM Length L Ch R = 1 ,1074.2  ,101.7,102.1,102.4
XS GIS Cut Line= 4
      1763543.94      196106.585     1763688.561      196309.055
     1763793.741      196501.008     1763906.809      196719.255
#Sta/Elev= 30
       0 1466.91    19.9 1455.31    39.8 1441.73    64.7 1426.53   124.4 1395.81
   164.2 1385.08     219 1375.06   253.8 1363.54   278.7 1352.42   288.6 1349.08
   303.5 1346.43   323.4 1345.33   343.4 1339.88   358.3 1337.75   358.4 1337.75
   363.2 1337.82   388.1 1346.26     418  1365.6   427.9 1370.23   497.2 1390.91
   511.9 1396.57   531.6 1401.93   546.4 1407.46     566 1418.37   590.6 1430.18
   615.2 1441.15   634.8 1447.59   664.3 1460.75   674.2 1466.54   713.5 1486.21
#Mann= 3 , 0 , 0
       0      .1       0   343.4    .045       0   358.4      .1       0
Bank Sta=343.4,358.4
XS Rating Curve= 0 ,0
Exp/Cntr=0.3,0.1

Type RM Length L Ch R = 1 ,972.1   ,64.6,64.2,63.9
XS GIS Cut Line= 3
     1763460.523       196092.37     1763656.196      196458.636
     1763839.913      196823.942
#Sta/Elev= 30
       0 1496.05    39.6 1470.54      89 1441.43   123.6 1424.41   222.5 1392.83
   252.1 1386.23     267 1384.71   281.8 1378.94   301.6 1373.25   316.4 1366.79
   336.2    1354   360.9 1339.81   365.8 1337.69   385.4 1333.95   395.5 1332.41
   400.4    1333   400.4 1333.01   420.2 1341.29   445.2 1349.54   465.1 1358.57
     510 1370.62   534.9 1382.02   554.9 1386.52   574.8 1393.54   644.6 1430.43
   669.6 1441.93   694.5 1455.12   709.5 1461.28   729.4 1473.69   824.2 1519.14
#Mann= 3 , 0 , 0
       0      .1       0   385.4    .045       0   400.4      .1       0
Bank Sta=385.4,400.4
XS Rating Curve= 0 ,0
Exp/Cntr=0.3,0.1

Type RM Length L Ch R = 1 ,907.9   ,153.8,147.8,141.9
XS GIS Cut Line= 4
     1763411.361      196215.813     1763549.356      196392.515
     1763631.817      196547.339     1763737.838      196769.478
#Sta/Elev= 30
       0 1453.37    39.9 1432.76    64.8 1421.28    79.7 1412.92    99.6 1406.58
   114.6 1396.98   124.6    1392   169.4 1378.19   229.1  1366.1   238.8 1362.42
   248.6 1357.18   263.2 1344.16   287.6 1333.45   295.7 1332.06   297.3 1331.98
   310.7 1333.66   331.4 1337.54   360.6 1346.57   399.6 1362.72     439 1368.34
   463.6 1374.49   478.4  1379.4   527.6 1404.33   532.5 1405.45   547.3 1413.97
   576.8 1427.81   586.7 1431.86   606.4 1436.46   621.1 1444.84   645.8 1454.94
#Mann= 3 , 0 , 0
       0      .1       0   295.7    .045       0   310.7      .1       0
Bank Sta=295.7,310.7
XS Rating Curve= 0 ,0
Exp/Cntr=0.3,0.1

Type RM Length L Ch R = 1 ,760     ,175.6,172.8,170.1
XS GIS Cut Line= 4
     1763286.828      196274.714     1763380.911        196437.9
       1763574.6       196641.58      1763645.28      196804.819
#Sta/Elev= 30
       0 1447.63    14.9    1437    44.6 1418.02    69.4 1403.61   104.1 1385.85
     114  1382.6   123.9 1380.71   148.7 1377.98   188.4 1375.45   203.2  1371.7
   222.9  1363.8   237.7 1355.08   247.5 1347.04   252.5 1342.13   257.4 1335.88
   267.3 1331.64   279.8 1329.78   282.1 1329.72   294.8 1332.06   311.6  1339.8
   346.2 1345.59     361 1346.58   380.7 1344.94   390.5 1346.25   415.2 1359.26
   425.1 1363.09   484.3 1377.35   573.2 1400.66   607.8 1415.82   647.3 1436.24
#Mann= 3 , 0 , 0
       0      .1       0   279.8    .045       0   294.8      .1       0
Bank Sta=279.8,294.8
XS Rating Curve= 0 ,0
Exp/Cntr=0.3,0.1

Type RM Length L Ch R = 1 ,587.3   ,63.3,67.9,72.6
XS GIS Cut Line= 4
     1763159.244      196426.419     1763280.358      196591.814
     1763485.721      196761.311      1763549.67      196889.209
#Sta/Elev= 30
       0 1407.78      15 1401.07      60 1388.66      80 1384.73     100 1382.14
     125 1377.81     150 1372.51     190  1359.2   214.9 1345.87   234.6 1334.17
   244.4 1331.37   260.7 1328.87   269.1  1329.1   275.7 1328.57   288.8 1327.88
   298.7  1328.9   313.5 1333.21   323.3 1335.34   367.7 1338.18   372.6 1339.04
   382.5 1343.23   392.4 1346.11   412.1 1346.85   426.9 1350.98   431.8 1352.91
   466.3 1370.82   505.8 1394.88   530.4 1411.05   555.1 1425.81   614.3 1457.83
#Mann= 3 , 0 , 0
       0      .1       0   260.7    .045       0   275.7      .1       0
Bank Sta=260.7,275.7
XS Rating Curve= 0 ,0
Exp/Cntr=0.3,0.1

Type RM Length L Ch R = 1 ,519.3   ,129.1,129.2,129.3
XS GIS Cut Line= 4
     1763063.857      196421.497     1763211.533      196592.027
      1763348.66      196764.315      1763484.03      196903.201
#Sta/Elev= 30
       0 1441.81    24.5 1425.87    53.9 1407.93    63.8 1402.92    83.4 1396.22
    93.2 1394.08   142.2 1391.97   156.9 1389.74   181.4 1381.07   215.8 1370.98
   230.5 1365.98     255 1359.33   269.6 1352.42   303.9 1330.11   308.8 1328.34
   323.4 1328.02     331 1328.11     346  1328.5   387.1 1331.97   411.5 1335.71
   450.8 1338.49   460.7  1342.1   475.6    1345   485.6 1349.23   525.4 1371.28
   560.2 1388.74     585  1403.7   604.9 1417.59   619.8 1426.54   639.7 1436.87
#Mann= 3 , 0 , 0
       0      .1       0     331    .045       0     346      .1       0
Bank Sta=331,346
XS Rating Curve= 0 ,0
Exp/Cntr=0.3,0.1

Type RM Length L Ch R = 1 ,390.2   ,152.9,155.1,157.2
XS GIS Cut Line= 4
     1762993.535      196507.641      1763123.63      196686.961
     1763244.935      196838.153     1763373.273        196957.7
#Sta/Elev= 30
       0 1422.78    24.6  1409.2    34.5 1404.83    44.3 1401.58    73.8 1396.01
   103.4 1393.07   132.9 1388.61   162.5 1382.38     192 1373.49   221.5    1362
   231.5 1356.77   256.3 1341.42   276.2 1332.36   286.2 1329.07   296.1 1327.26
   300.8 1327.34   315.8 1328.91   340.8 1328.25   355.7 1328.88   365.7 1330.82
   380.6 1340.41   405.4 1351.47   420.2 1355.26   459.2 1361.29   478.7 1371.13
   512.8 1385.42   532.3 1392.72   546.9 1399.95   561.5 1403.91   590.8 1413.62
#Mann= 3 , 0 , 0
       0      .1       0   300.8    .045       0   315.8      .1       0
Bank Sta=300.8,315.8
XS Rating Curve= 0 ,0
Exp/Cntr=0.3,0.1

Type RM Length L Ch R = 1 ,235.1   ,183.8,187.4,194.2
XS GIS Cut Line= 4
     1762898.601      196604.333     1762998.809      196757.283
      1763106.05      196920.781     1763220.323       197029.78
#Sta/Elev= 30
       0 1401.64     9.9 1394.92    24.7 1386.36    39.5 1379.17    54.4 1373.49
    64.2 1371.09      89 1369.25   148.3  1361.6   153.2 1360.42   163.1 1355.95
   192.6 1338.43   207.3 1332.69   212.2 1331.64   241.5  1329.5     266 1323.02
   280.6 1323.18   293.7 1321.21   295.3 1320.95   300.2 1320.95   308.7 1322.84
   319.7 1326.56     349 1344.01   363.7 1350.08   388.2 1358.02   412.9 1364.07
   427.7 1366.66   462.3 1377.03   496.8 1392.56   521.5 1405.51   536.3  1412.4
#Mann= 3 , 0 , 0
       0      .1       0   293.7    .045       0   308.7      .1       0
Bank Sta=293.7,308.7
XS Rating Curve= 0 ,0
Exp/Cntr=0.3,0.1

Type RM Length L Ch R = 1 ,47.7    ,75.6,47.7,16.5
XS GIS Cut Line= 4
     1762777.735      196658.833     1762855.089      196843.427
     1762928.927      197005.168     1763027.377      197100.102
#Sta/Elev= 30
       0 1411.34    14.6 1401.72    48.8 1380.62    68.3 1370.18    97.6 1359.12
   102.5 1356.96   112.3 1350.79   117.2 1348.95   141.6 1345.63   146.4 1343.93
     166 1332.05   175.7 1327.21   180.6 1325.62   190.4 1323.97   219.9 1323.23
   254.5 1320.49   262.8 1318.74   269.3 1317.68   277.8 1318.25     289 1320.41
   313.7 1322.37   323.6 1324.16   328.6 1326.39   353.2  1341.3     373 1349.12
   402.4 1358.65   426.8  1368.7   456.1  1382.8   500.1  1406.4   514.7 1413.12
#Mann= 3 , 0 , 0
       0      .1       0   262.8    .045       0   277.8      .1       0
Bank Sta=262.8,277.8
XS Rating Curve= 0 ,0
Exp/Cntr=0.3,0.1

Chan Stop Cuts=-1
Use User Specified Reach Order=0
